HEC-RAS study RBNSONFRK.prj: RBNSONFRK

--- RBNSONFRK.g01 (geometry) --- (continued)

Type RM Length L Ch R = 1 ,25291.2 ,191.2,190.4,191.8
XS GIS Cut Line= 4
     1662893.832      315075.471      1663032.72      315209.151
     1663301.818      315549.429      1663461.54      315789.012
#Sta/Elev= 30
       0  994.99    38.6  980.96    48.2  976.39    77.1  959.24   115.7  935.56
   163.9   904.9   221.7  867.07     241  855.27   250.6  851.63   260.2  850.35
   269.9  849.56   279.5  848.13   308.5  842.69   322.9  841.16   327.7  840.89
   337.9  841.23   375.9  843.13   501.3  847.83   530.2  850.94     588   855.4
   597.7  856.41   607.3  858.26     617  861.64   626.6  866.04     665  884.93
   751.4  928.43   799.4  951.16     809  955.29   828.2  962.52   914.5  991.24
#Mann= 3 , 0 , 0
       0     .08       0   322.9    .045       0   337.9     .06       0
Bank Sta=322.9,337.9
XS Rating Curve= 0 ,0
Exp/Cntr=0.3,0.1

Type RM Length L Ch R = 1 ,25100.8 ,305.4,314.3,321.7
XS GIS Cut Line= 2
     1662909.585      315298.864     1663130.939      315669.957
#Sta/Elev= 30
       0  876.26     9.8   865.6    19.6  858.53    29.5  857.92    39.3  857.66
    49.1  856.48    58.9  853.73    68.7  850.07    78.6  846.74    88.4  844.79
    98.2  843.42     108  842.62   117.8  842.12   137.5  841.98   157.1  841.99
     167  841.72   186.6  840.79   192.2  840.65   196.4  840.55   207.2  840.77
   304.4  846.18   314.2  846.81   324.1  847.79   333.9  849.19     383  856.68
   392.8  858.48   402.6  860.47   412.5   863.2   422.3  866.27   432.1  870.26
#Mann= 3 , 0 , 0
       0     .08       0   192.2    .045       0   207.2     .08       0
Bank Sta=192.2,207.2
XS Rating Curve= 0 ,0
Exp/Cntr=0.3,0.1

Type RM Length L Ch R = 1 ,24786.6 ,423.3,437.6,452.7
XS GIS Cut Line= 3
     1662731.634      315346.607     1662838.276      315864.533
     1663205.005       316315.97
#Sta/Elev= 30
       0  861.32    29.4  854.88      49  851.29   107.7  843.02   156.7  842.49
   264.4  842.96   313.4  841.71     346  839.49   352.5  839.22     361  839.29
   411.3  841.14   421.1  842.28   450.4  849.67     470  855.71   489.6  863.18
   528.8  879.94   548.2  889.39   654.8  955.18   674.2  965.48   732.4  994.68
   780.8 1021.68   809.9 1036.87   829.3 1045.88   906.8 1073.04   926.2 1081.32
   955.3 1098.22   994.1 1122.51  1023.2 1138.54    1062 1156.96  1110.4 1176.39
#Mann= 3 , 0 , 0
       0     .06       0     346    .045       0     361     .08       0
Bank Sta=346,361
XS Rating Curve= 0 ,0
Exp/Cntr=0.3,0.1

Type RM Length L Ch R = 1 ,24349   ,587.3,592,596.5
XS GIS Cut Line= 3
     1662722.953      315140.443     1662371.391      315802.336
     1662197.779      315971.607
#Sta/Elev= 30
       0  951.48   136.3  871.46     146  867.23   165.5  863.95   175.2  860.12
   184.9   855.3   194.7  851.75   204.4  849.93   272.5  843.26   330.9   839.2
   360.1   838.1   381.9  838.12   396.9   838.8   418.5  843.95   428.3  843.82
   476.9   840.2   506.1  839.35   622.9   839.6   671.6  841.29   691.1  842.94
   739.7  848.73   788.3  858.71     798  861.02   807.7  864.22   836.8  876.45
   846.4   881.5   875.6  899.51   914.4   924.6     924  930.36   991.9  966.81
#Mann= 3 , 0 , 0
       0     .06       0   381.9    .045       0   396.9     .06       0
Bank Sta=381.9,396.9
XS Rating Curve= 0 ,0
Exp/Cntr=0.3,0.1

Type RM Length L Ch R = 1 ,23757   ,380.6,377.8,374.4
XS GIS Cut Line= 3
     1662469.047      315003.725     1662084.932      315492.006
     1661976.425      315546.259
#Sta/Elev= 30
       0  930.27      68  894.48   106.8  873.47   116.5  868.43   126.2  864.39
   135.9  862.12   145.6  861.48   155.3  860.36     165  858.39   174.7  855.92
   184.4  852.95   203.8  846.21   213.6  843.22   223.3  841.15   242.7  839.71
   252.4   839.3   281.5   838.8   359.2   839.3     398   839.1   475.6  839.37
   495.1  839.19   533.9  838.15   543.6   838.1   566.2   838.1   581.2  838.46
   592.1  840.05   611.6   845.2   621.3  848.38   630.6  853.11   742.6  912.38
#Mann= 3 , 0 , 0
       0     .06       0   566.2    .045       0   581.2      .1       0
Bank Sta=566.2,581.2
XS Rating Curve= 0 ,0
Exp/Cntr=0.3,0.1

Type RM Length L Ch R = 1 ,23379.2 ,96.8,94.8,93.6
XS GIS Cut Line= 4
     1662456.176       314841.76     1662017.964      314979.117
     1661863.884      315222.172     1662092.779      316157.147
#Sta/Elev= 30
       0  982.27     127  929.49   166.1  911.36   224.7  882.22   244.3  873.84
     254   871.6   293.1  867.14   390.8  857.76   429.9  855.89   468.8  848.86
   507.2  847.87   555.2  840.46   612.7   838.1   629.7  838.12   644.7  838.93
   708.6  844.69   796.1  874.02   933.6  906.45  1041.7   920.2  1090.8  925.03
  1130.1  926.81  1208.7  927.59  1257.8   937.4  1306.9  944.26    1356  957.97
  1414.9  969.69  1473.9  979.67  1581.9 1005.98  1640.8 1026.34  1709.6 1055.72
#Mann= 3 , 0 , 0
       0     .06       0   629.7    .045       0   644.7      .1       0
Bank Sta=629.7,644.7
XS Rating Curve= 0 ,0
Exp/Cntr=0.3,0.1

Type RM Length L Ch R = 1 ,23284.3 ,319.6,290.6,261.1
XS GIS Cut Line= 3
     1662065.707      314638.405     1661777.078      315217.832
     1661859.387      315395.146
#Sta/Elev= 30
       0  938.39    39.2   917.6   107.9  883.42   117.7     879   137.3  872.57
   166.7  865.14   186.4  861.42   245.2     852   274.6  848.67   294.2  847.55
   372.7  841.51   382.5  841.28   411.9  842.01   421.8  841.26   441.4  838.68
   478.2  837.65   480.6  837.64   493.2   838.2     510  839.06   529.6   838.6
   539.4  839.05   578.7  841.96   627.7  846.98   657.1  849.41   666.9  852.06
     706  868.97   803.7  908.04   813.5  911.55   823.3  914.26   842.8  918.54
#Mann= 3 , 0 , 0
       0     .06       0   478.2    .045       0   493.2     .06       0
Bank Sta=478.2,493.2
XS Rating Curve= 0 ,0
Exp/Cntr=0.3,0.1

Type RM Length L Ch R = 1 ,22993.7 ,748.3,738.4,726.7
XS GIS Cut Line= 4
     1660609.519      314630.206     1661225.863      314835.887
     1661724.995      315319.828     1661907.262      315506.942
#Sta/Elev= 30
       0 1149.24    38.8 1131.16    87.3 1106.26   126.1 1084.92   242.4 1018.28
   339.4  966.19   407.3   931.3   475.2  898.18   484.9  894.01   494.6  891.05
   543.1  879.28   601.3  863.76   649.8  855.04   728.1  850.34  1188.3  839.81
  1248.2  835.99  1256.8  835.79  1263.2  837.07  1266.6  837.75    1296  852.14
  1315.6  855.45  1325.4  858.72    1374  889.38  1393.4  900.71  1412.7  910.03
    1432  917.62  1461.1  922.94  1490.1  926.09  1557.8  928.82  1606.2  927.45
#Mann= 3 , 0 , 0
       0     .06       0  1248.2    .045       0  1263.2     .06       0
Bank Sta=1248.2,1263.2
XS Rating Curve= 0 ,0
Exp/Cntr=0.3,0.1

Type RM Length L Ch R = 1 ,22255.3 ,415.7,427,437.5
XS GIS Cut Line= 2
     1660828.422      315537.579     1661729.029      315902.162
#Sta/Elev= 30
       0  859.92    19.6  859.69    78.5  857.81     265  847.84   431.8  840.81
   549.6     835   568.7   834.7   583.7  834.82   588.8  834.94   618.3  837.79
   637.9  838.95   667.4  839.79   716.4  840.35   736.1  841.26   745.9  843.19
   765.5  850.63   775.3  853.67     795  856.24   804.8  859.45   814.6  865.82
   824.4  874.25   834.2  882.02     844  888.59   853.8  894.78   873.5  905.43
   883.3  910.14   902.9  918.55   912.7  922.14   942.2  931.65   971.6  942.96
#Mann= 3 , 0 , 0
       0     .06       0   568.7    .045       0   583.7     .06       0
Bank Sta=568.7,583.7
XS Rating Curve= 0 ,0
Exp/Cntr=0.3,0.1

Type RM Length L Ch R = 1 ,21828.3 ,163.4,165.2,167.1
XS GIS Cut Line= 2
     1660730.766      315589.662     1661444.741      316294.957
#Sta/Elev= 30
       0  859.89    78.7  857.33    88.6  856.78   118.1  853.68   127.9  852.98
   196.8  850.05   255.8  848.17   275.5  848.05   344.4  846.96   511.6   841.6
   619.9     840   659.2  838.46   718.3  834.74   721.9  834.74   728.1  834.74
   736.9  835.59   737.9  835.69   747.8  839.16   757.6  843.58   767.4  846.17
   777.3  847.21   787.1  850.03     797  856.15   816.6  870.73   836.3  885.81
   846.2  892.49     856  897.83     915  925.16   964.2  947.25  1003.6  964.58
#Mann= 3 , 0 , 0
       0     .06       0   721.9    .045       0   736.9      .1       0
Bank Sta=721.9,736.9
XS Rating Curve= 0 ,0
Exp/Cntr=0.3,0.1

Type RM Length L Ch R = 1 ,21663   ,63.6,63.6,63.6
XS GIS Cut Line= 2
     1660225.273      315162.941      1661436.21      316571.361
#Sta/Elev= 30
       0   956.1    78.6  927.28   117.9  914.44   216.2  887.29   255.5  880.26
   412.8  871.63   540.5  866.88     629  861.55   707.6  861.18   746.9  857.87
     855  855.53   982.8  848.17  1051.6  845.53  1228.4  843.59  1346.4  839.25
  1380.3  834.78  1385.7  834.53  1395.3  836.15  1415.2  845.27  1434.8  848.61
  1444.7  852.35  1454.5  859.88    1484  886.23  1493.8  893.25  1542.9  914.54
  1641.2  961.35  1700.2   986.5  1739.5   997.4  1778.8  1010.5  1857.4 1040.67
#Mann= 3 , 0 , 0
       0     .06       0  1380.3    .045       0  1395.3      .1       0
Bank Sta=1380.3,1395.3
XS Rating Curve= 0 ,0
Exp/Cntr=0.3,0.1

Type RM Length L Ch R = 1 ,21599.5 ,225.6,221.8,217.8
XS GIS Cut Line= 3
     1659990.898       316089.59     1660790.418      315917.367
     1661386.297      316610.424
#Sta/Elev= 30
       0  1117.4    77.9 1084.49   126.6 1065.92   214.2 1026.96   360.2  973.77
   486.8     914   593.9  865.16   613.4  857.44   623.1  854.91   642.6  852.37
   681.6  851.24   749.7   850.6   798.4  851.86   906.3  845.18  1132.4  841.81
  1201.2  838.77  1252.2  834.24  1260.1  834.05  1267.2  835.57  1289.6   845.9
  1309.3  849.84  1319.1  853.37  1368.2  891.01    1378  894.73  1397.7  897.91
  1417.4  904.77  1515.6  953.74  1535.3  962.16  1623.8  996.06  1731.9 1025.28
#Mann= 3 , 0 , 0
       0     .06       0  1252.2    .045       0  1267.2      .1       0
Bank Sta=1252.2,1267.2
XS Rating Curve= 0 ,0
Exp/Cntr=0.3,0.1

Type RM Length L Ch R = 1 ,21377.7 ,213.4,205.2,196.9
XS GIS Cut Line= 4
     1660342.311      316162.579     1660622.259      316153.898
     1660930.418      316407.804     1661162.623      316503.291
#Sta/Elev= 30
       0  975.51    86.9  927.77   106.2  918.06   183.5  884.79   270.4  851.45
   280.1  848.61   289.8  847.31   299.6  846.68     358  843.68   387.2  842.63
   426.2  842.06   513.8  842.34   552.8  841.24     582  839.25     633  833.93
   640.4  833.75     648  834.38   650.2  834.56     689  842.88   708.3  845.04
     718  846.94     747  855.69   756.6  859.96   814.6  888.73   824.2   893.1
   833.9  896.72   862.8  906.22   911.1     921   920.8   924.8   930.4  929.42
#Mann= 3 , 0 , 0
       0     .06       0     633    .045       0     648      .1       0
Bank Sta=633,648
XS Rating Curve= 0 ,0
Exp/Cntr=0.3,0.1

Type RM Length L Ch R = 1 ,21172.6 ,392.3,394.1,395.2
XS GIS Cut Line= 2
     1659975.839      316268.227     1661178.096      316687.498
#Sta/Elev= 30
       0 1114.05    88.2 1087.93   107.7 1081.59   127.3 1073.18   205.7 1035.13
   225.3 1027.25   313.4  994.26     333  984.44     431  927.74   450.5  917.35
   538.7   881.1   626.8  846.78   636.6  844.63   656.2  842.93     715  840.31
     764  839.11   842.3  832.89   843.8  832.93   852.1  833.15   858.8  834.11
   881.5  838.74   920.7   840.8   940.3  842.51     950  844.39   969.6  849.77
     999  859.03  1087.2  893.15  1126.4  903.94  1175.3  923.25  1273.3  953.54
#Mann= 3 , 0 , 0
       0     .06       0   843.8    .045       0   858.8     .06       0
Bank Sta=843.8,858.8
XS Rating Curve= 0 ,0
Exp/Cntr=0.3,0.1

Type RM Length L Ch R = 1 ,20778.5 ,262,268.2,274.4
XS GIS Cut Line= 3
     1660149.474      316621.912      1660720.22      316873.648
     1661091.314      317016.877
#Sta/Elev= 30
       0  993.29     9.8  990.26    19.5  986.04    68.2   962.2   204.7  898.31
   224.2  888.02   272.9  860.25   302.2  845.42   321.6  837.14   331.4  833.93
   340.8  832.32   341.1  832.27   355.8  832.77   370.4  833.78   399.6  834.67
   438.6  834.04   448.4   834.5   506.8  837.98   584.8  845.76   672.3  848.46
   740.2  853.89   759.6  856.87   817.8  869.14   846.9  873.59   866.3  875.81
   885.8  877.28     944  879.37   963.4  883.65   973.1   886.4  1021.6  902.18
#Mann= 3 , 0 , 0
       0      .1       0   340.8    .045       0   355.8     .08       0
Bank Sta=340.8,355.8
XS Rating Curve= 0 ,0
Exp/Cntr=0.3,0.1

Type RM Length L Ch R = 1 ,20510.3 ,208.2,212,215.5
XS GIS Cut Line= 2
     1660158.719      316851.035      1660702.99      317298.952
#Sta/Elev= 30
       0  934.23    39.2  913.12    78.3   891.7   127.3  865.51   166.4  844.11
   176.2  839.75     186  836.97   210.3  833.07   215.4  832.43   225.2  832.15
   225.3  832.16     235  832.81   274.1  837.16   303.5  839.95   332.9  842.06
   352.4  842.81   450.3  843.49   538.4   841.7   567.8   841.6   577.6  841.92
   587.4  843.46   597.2  846.06     607  849.02   616.8  850.66   626.6  851.34
   636.4  852.44   646.1  854.53   665.7  859.46   695.1  866.05   704.9  868.64
#Mann= 3 , 0 , 0
       0      .1       0   210.3    .045       0   225.3     .06       0
Bank Sta=210.3,225.3
XS Rating Curve= 0 ,0
Exp/Cntr=0.3,0.1

Type RM Length L Ch R = 1 ,20298.4 ,599.1,608.4,618
XS GIS Cut Line= 2
     1659902.054      316830.727     1661004.485       317967.88
#Sta/Elev= 30
       0 1020.82    68.9  994.23   216.4  918.61   245.9   904.3   383.7  844.08
   393.5  840.31   403.3  837.76   471.5  831.52   472.2  831.49   486.5  832.28
   521.4  835.43   600.1  839.84   668.9  840.49   747.6  843.62   806.7  848.69
   875.5  856.22     905  858.16   914.9   860.4   924.7  864.03   973.9  886.05
  1062.4  911.15  1111.6  928.58  1170.6  950.93    1210  961.73  1278.9  984.99
  1426.4 1028.86  1475.6 1042.52  1534.6 1061.03  1564.1 1067.86  1583.8 1068.82
#Mann= 3 , 0 , 0
       0     .06       0   471.5    .045       0   486.5     .06       0
Bank Sta=471.5,486.5
XS Rating Curve= 0 ,0
Exp/Cntr=0.3,0.1

Type RM Length L Ch R = 1 ,19689.9 ,304.6,305.8,310.8
XS GIS Cut Line= 3
     1659745.523      317173.864     1659910.453      317699.037
     1660081.894      317892.179
#Sta/Elev= 30
       0  906.11   167.1  840.53   176.9  837.61   186.8  836.32   245.7   834.7
   275.2  834.17   314.6   834.4     344  833.85   363.7  832.77   383.4  831.24
     403  829.29   415.6  828.71   422.7  828.61   430.6  828.73   442.3  829.63
   491.5  835.77     521  838.38     560  840.76   617.4  843.01   636.6  844.06
   646.1  845.81   655.7  848.78   665.2  851.15   674.8  851.99   684.4  853.92
   693.9  858.57   703.5   864.2   713.1  869.27   722.6  873.84   808.7  913.39
#Mann= 3 , 0 , 0
       0     .06       0   415.6    .045       0   430.6     .06       0
Bank Sta=415.6,430.6
XS Rating Curve= 0 ,0
Exp/Cntr=0.3,0.1

Type RM Length L Ch R = 1 ,19384.1 ,201.7,210.4,214.8
XS GIS Cut Line= 3
     1659578.703      317150.605     1659613.426      317805.987
     1659552.662      318587.237
#Sta/Elev= 30
       0  924.93    19.6  916.37   235.1  837.82   244.9  835.84   264.5  833.84
   350.6  828.21   352.6  828.17   365.6  828.32   617.1  835.19   646.5  836.51
   656.3  837.99   666.1  841.33   685.7  854.48   695.5  859.69   715.1  863.74
   724.9  868.22     862  953.43   881.6  964.35   930.6  985.83     960  996.24
  1018.7 1014.32  1067.7 1027.65  1087.3 1032.28  1116.7 1037.44  1146.1 1044.85
  1185.2 1050.84  1253.8 1064.96  1332.2  1078.8  1371.3  1083.6  1439.9 1089.07
#Mann= 3 , 0 , 0
       0     .06       0   350.6    .045       0   365.6     .06       0
Bank Sta=350.6,365.6
XS Rating Curve= 0 ,0
Exp/Cntr=0.3,0.1

Type RM Length L Ch R = 1 ,19173.7 ,415.7,411.2,406.3
XS GIS Cut Line= 2
     1659435.193      317217.266     1659365.748      317948.603
#Sta/Elev= 30
       0  901.98    19.6  895.15    68.6  876.68   156.7  844.23   166.5  841.54
   176.3  841.11   186.1  839.31   195.9  833.37   202.5  829.86   205.7  828.16
   215.5   827.9   217.5  827.94   264.5  828.88   362.4   829.2   401.6   829.7
   460.4  831.26   509.3  833.55   519.1  834.23   528.9  837.27   538.7  843.46
   558.3  857.77   568.1   863.8   577.9  867.02   587.7  868.41   597.5  870.98
   607.3  875.34   646.5  895.42   675.9  911.01   705.2   927.3   734.6  943.98
#Mann= 3 , 0 , 0
       0      .1       0   202.5    .045       0   217.5     .06       0
Bank Sta=202.5,217.5
XS Rating Curve= 0 ,0
Exp/Cntr=0.3,0.1

Type RM Length L Ch R = 1 ,18762.5 ,100.5,88,75.8
XS GIS Cut Line= 4
     1659062.234      317153.596     1659075.636      317346.699
     1659119.703      317774.148     1659198.953      317889.273
#Sta/Elev= 30
       0  880.36    38.7  872.01    96.8  857.43   116.1  853.31   135.5  850.42
   174.2  846.66   193.6  842.85   203.3  841.99   222.9   841.7   242.4  840.52
   291.2  835.16   330.3   832.5   379.1  832.25   437.7  827.77   476.8  826.45
   496.3  826.21   497.9  826.21   512.9  826.38   525.6  827.32   545.2  830.15
   554.9  832.11   564.7  835.49   641.9  869.29   651.2  872.41   669.9  874.64
   679.2  876.83   688.5  880.37   735.1  902.82   744.4  906.28     763  912.13
#Mann= 3 , 0 , 0
       0      .1       0   497.9    .045       0   512.9     .06       0
Bank Sta=497.9,512.9
XS Rating Curve= 0 ,0
Exp/Cntr=0.3,0.1

Type RM Length L Ch R = 1 ,18674.5 ,483.5,473,464
XS GIS Cut Line= 3
     1658592.779      317250.897     1658834.966      317435.792
     1659308.925      318068.605
#Sta/Elev= 30
       0 1020.56    29.5 1008.64    39.3 1004.23   157.3  944.05   167.1   937.7
   206.4  905.83   226.1  890.97   294.9  842.17   304.7  836.94   314.5  835.09
   324.2  834.73   568.2  831.08   597.5  829.42   624.9  826.91   636.6  826.34
   639.9  826.56   646.3  826.99   656.1  828.61   665.8  830.64   675.6  833.43
   763.5  869.81   773.2  872.76   792.7  875.37   802.5   878.5   841.5  897.38
   851.3  901.49   929.4  925.21     988  944.86  1056.3  972.62  1095.3  989.44
#Mann= 3 , 0 , 0
       0     .06       0   624.9    .045       0   639.9      .1       0
Bank Sta=624.9,639.9
XS Rating Curve= 0 ,0
Exp/Cntr=0.3,0.1

Type RM Length L Ch R = 1 ,18201.4 ,289.7,295.4,298.9
XS GIS Cut Line= 2
      1658454.29      317863.968     1658977.293      318195.999
#Sta/Elev= 30
       0  911.26      59  888.24    78.7  880.15   108.2  865.48   157.3  840.61
   167.2   836.2     177  833.48   186.8  832.18   226.2  829.12   255.7  826.53
   265.5  826.61   269.1  827.15   275.3  828.08   284.1  830.05     295  832.42
   304.8  833.55   324.5  835.28   383.5  841.12   432.7  844.39   462.2  847.51
     472  849.05   481.8  851.57   491.7  854.68   501.5  858.26   511.3  862.35
   521.2  865.88     531  867.37   540.8  868.24   550.7  870.13   619.5  891.65
#Mann= 3 , 0 , 0
       0     .06       0   269.1    .045       0   284.1      .1       0
Bank Sta=269.1,284.1
XS Rating Curve= 0 ,0
Exp/Cntr=0.3,0.1

Type RM Length L Ch R = 1 ,17906.1 ,336.4,347.7,358.9
XS GIS Cut Line= 2
     1658333.044      318070.744     1659144.676      318773.869
#Sta/Elev= 30
       0  882.16     9.8  879.31    29.3  872.75    48.8  865.37    97.6  843.04
   107.4  839.36   117.2  837.63   156.2  835.22   185.5  832.81   235.9  826.76
     244  826.69   250.9  827.63   273.3   831.5   341.7  835.85   380.7  839.03
   458.8  848.57   488.1  853.68   507.6  855.93   517.4  859.02   566.2  882.32
     576  886.85   585.7  890.64   605.2   896.5   722.4  929.76     781  950.96
   859.1  980.23   927.4 1009.33   956.7 1021.09  1054.3 1055.05  1073.8 1060.95
#Mann= 3 , 0 , 0
       0     .06       0   235.9    .045       0   250.9     .06       0
Bank Sta=235.9,250.9
XS Rating Curve= 0 ,0
Exp/Cntr=0.3,0.1

Type RM Length L Ch R = 1 ,17558.3 ,65.4,65.4,65.4
XS GIS Cut Line= 2
     1658126.315      318108.253     1658470.065       319024.92
#Sta/Elev= 30
       0  885.95    19.6  883.96    68.5  875.74   156.6  867.77   166.4  865.24
   176.2  860.88   205.6  843.38   215.4   838.9   225.2  837.15   313.3  833.17
   332.9  831.22   360.4   826.4   362.2  826.12   375.4  826.89   401.4  832.13
   430.8     835   460.1  836.13   479.7  838.23   538.4  840.88   675.5  842.08
   685.3  841.27   704.9   837.7   724.5  836.69   763.6  840.28   812.6  842.52
   822.4  845.33   851.7  857.08   939.8  884.24   959.4  888.69     979  891.73
#Mann= 3 , 0 , 0
       0     .06       0   360.4    .045       0   375.4     .06       0
Bank Sta=360.4,375.4
XS Rating Curve= 0 ,0
Exp/Cntr=0.3,0.1

Type RM Length L Ch R = 1 ,17493   ,161.6,156.6,151.5
XS GIS Cut Line= 2
     1658067.287      318136.031     1658411.037      319052.698
#Sta/Elev= 30
       0  869.97    19.6     871    68.5  877.22    97.9  875.65   146.8  870.64
   166.4  867.54   176.2  863.92   215.4   841.2   225.2  836.55     235  834.55
   332.9  829.86   361.7  825.79   362.2  825.72     372  826.17   376.7  827.34
   391.6  831.31     421  833.91   499.3   835.6   587.4  832.98   616.8  834.38
   636.4  836.31   675.5   841.7   685.3  842.34   704.9  841.82   714.7  843.22
   734.2  850.57   783.2  865.14   851.7  891.85   939.8  914.82     979  921.28
#Mann= 3 , 0 , 0
       0     .06       0   361.7    .045       0   376.7     .06       0
#XS Ineff= 2 , 0
                          498.59          836.03
Permanent Ineff=
       F       F
Bank Sta=361.7,376.7
XS Rating Curve= 0 ,0
Exp/Cntr=0.3,0.1

Type RM Length L Ch R = 1 ,17336.4 ,176.1,174.6,173
XS GIS Cut Line= 3
      1657903.38      317748.214     1657966.314      318394.915
     1658343.328      318988.462
#Sta/Elev= 30
       0  899.26    48.5  885.68   135.8  867.44     194  858.58   271.5  849.36
   310.3  842.53   378.2  838.08   475.2  836.62   523.7   839.6   533.4   840.5
   552.8  844.28   581.9  845.83   630.4  842.68   659.5  839.06   669.3  837.33
   698.6  829.68   708.4   828.1   737.6  826.25   794.6  824.22   796.2  824.19
   809.6  824.46   913.4  829.92  1001.3  832.48  1040.4  837.35  1118.5  838.98
  1147.8  843.81  1167.4   845.4  1186.9   851.3  1284.6  891.32  1352.9  908.62
#Mann= 3 , 0 , 0
       0     .06       0   794.6    .045       0   809.6     .06       0
Bank Sta=794.6,809.6
XS Rating Curve= 0 ,0
Exp/Cntr=0.3,0.1

Type RM Length L Ch R = 1 ,17161.8 ,848.6,852.8,856.9
XS GIS Cut Line= 3
     1657334.804      317928.335     1657775.342      318431.808
     1658218.328      319013.635
#Sta/Elev= 30
       0  906.21    68.9   898.9   177.1     877   226.3  869.58   275.5  860.38
     305  858.47   383.7  857.51   482.1  859.79   560.8  855.39   570.6  854.44
   619.8  842.57     669  834.94   717.8   832.6   795.8  831.22   851.8  824.26
   854.2  824.05   866.8  824.32     942  829.02   990.8  829.77  1117.5  828.43
  1166.3  829.58  1195.5  831.88  1205.3  835.77    1215  841.56  1224.8  845.85
  1234.5  847.78    1254  849.44  1263.8  852.44  1341.8   891.3  1400.3  911.59
#Mann= 3 , 0 , 0
       0     .06       0   851.8    .045       0   866.8     .06       0
Bank Sta=851.8,866.8
XS Rating Curve= 0 ,0
Exp/Cntr=0.3,0.1

Type RM Length L Ch R = 1 ,16309   ,299.1,288.6,278.6
XS GIS Cut Line= 3
     1657051.948      318481.243     1657150.342      318583.717
     1657456.026      319172.561
#Sta/Elev= 30
       0  907.31    47.4  890.29    66.3  882.88   132.6   854.1   151.8   846.7
   190.8  835.13   239.6   824.3   249.4  822.77   259.2  822.96   288.4  825.31
   327.4  827.06   366.5  827.93   405.5  828.01   454.3  826.96   483.6  825.18
     511  822.87   512.8  822.74     526  823.16   551.8  826.27   581.1  828.12
   590.9  829.39   600.6   832.3   610.4  837.62   629.9  850.97   639.7  855.17
   659.2  859.17   668.9  862.91   717.7  890.04   737.2  898.68   805.5  927.04
#Mann= 3 , 0 , 0
       0     .06       0     511    .045       0     526     .08       0
Bank Sta=511,526
XS Rating Curve= 0 ,0
Exp/Cntr=0.3,0.1

Type RM Length L Ch R = 1 ,16020.4 ,384.8,389.2,392.8
XS GIS Cut Line= 2
     1656823.392      318684.693     1657326.099      319311.196
#Sta/Elev= 30
       0  923.12    19.6  913.84      49  898.73   146.9  845.24   166.5  835.43
   176.3  831.43   186.1   828.9   225.3  822.96   235.1  822.22   284.1  823.28
   347.7   821.4   352.6  821.34   362.7  821.41   391.8  825.98   401.6     827
   460.4  829.07   489.8  830.61   509.4  832.45   519.2  834.38     529  837.92
   538.8  843.03   548.6  847.07   568.2  850.45     578  854.15   626.9  883.18
   636.7  888.65   646.5  892.94   675.9  902.74   744.5  924.09   803.3  940.48
#Mann= 3 , 0 , 0
       0     .06       0   347.7    .045       0   362.7     .06       0
Bank Sta=347.7,362.7
XS Rating Curve= 0 ,0
Exp/Cntr=0.3,0.1

Type RM Length L Ch R = 1 ,15631.2 ,600.4,583.1,566.2
XS GIS Cut Line= 3
     1656468.918      318798.561     1656578.381      318925.564
     1656930.852       319302.77
#Sta/Elev= 30
       0   984.4    37.3  972.04    46.6   967.6    65.2  957.95    83.8  948.82
    93.2  944.88   130.4  931.03   139.7  927.29   158.4  919.11   206.6  897.09
   216.4  891.96   226.1  885.83   265.1  859.28   274.8  852.84   284.6  846.86
   294.3   841.6   313.8  831.84   323.5  826.57   333.3  822.24     343  821.32
   343.3  821.34   358.3  822.75   372.2  823.98   489.1  827.58   498.8  828.37
   547.6  834.22     567  835.94   586.5  837.24     606  838.12   683.9   840.1
#Mann= 3 , 0 , 0
       0      .1       0   343.3    .045       0   358.3     .06       0
Bank Sta=343.3,358.3
XS Rating Curve= 0 ,0
Exp/Cntr=0.3,0.1

Type RM Length L Ch R = 1 ,15048.1 ,489.4,492,493.9
XS GIS Cut Line= 3
     1655924.214      319460.453     1656274.601      319497.499
     1656896.436      319545.089
#Sta/Elev= 30
       0 1046.59    58.7 1011.75   166.4  954.74   176.2  950.31     186  946.84
   244.7  929.08   254.5  925.32   264.3  920.45   342.6  875.86   362.1  862.83
   410.8  825.17   420.6  820.14   425.7  819.34   430.3  818.62   440.7  819.09
   469.3  821.21   547.2  823.12   605.7  823.72   703.2   823.4   761.6  824.57
   810.3  826.35   820.1  828.06   839.6  834.32   859.1  838.07   868.8  843.59
   878.6  850.55   888.3  856.01     898  860.02   927.3  870.87     976  886.02
#Mann= 3 , 0 , 0
       0      .1       0   425.7    .045       0   440.7     .06       0
Bank Sta=425.7,440.7
XS Rating Curve= 0 ,0
Exp/Cntr=0.3,0.1

Type RM Length L Ch R = 1 ,14556.1 ,395.1,405.4,413.8
XS GIS Cut Line= 2
     1656236.689      319955.293     1656844.328       320059.46
#Sta/Elev= 30
       0  908.04     9.8  903.99    19.6  898.88    48.9  880.31    88.1   856.8
    97.9  849.93   107.6  841.81   117.4  832.95   127.2  824.88     137  819.38
   146.8  816.85   156.6  816.05   164.6  815.88   166.4  815.84   179.6  816.11
   185.9  816.52   205.5  819.35   215.3  820.02     274  820.78   332.7  820.34
   342.5  821.22   362.1   826.8   381.6  830.52   391.4  835.86   401.2  844.03
     411   851.5   430.6  863.46   450.1  874.67   567.6   929.6   616.5  952.02
#Mann= 3 , 0 , 0
       0      .1       0   164.6    .045       0   179.6     .06       0
Bank Sta=164.6,179.6
XS Rating Curve= 0 ,0
Exp/Cntr=0.3,0.1

Type RM Length L Ch R = 1 ,14150.6 ,532.8,543.7,554.6
XS GIS Cut Line= 2
     1656108.675      320222.172     1656529.377      320487.666
#Sta/Elev= 30
       0  903.87     9.8  900.74    19.5  896.59    29.3  891.71    58.5  876.05
      78  865.73   107.3  850.36   126.8  840.33   146.3  829.92   156.1  824.81
   165.8  820.98   175.6   819.2   224.4     817   234.1  816.42   245.8  815.92
   253.6  815.77   260.8  815.98   263.4  816.05   273.1  816.94   282.9  818.18
   292.6  819.22   341.4  824.05   409.7  831.52   419.4   832.4   438.9  832.99
   448.7  833.77   458.4  835.17     478  838.66   487.7     840   497.5  840.96
#Mann= 3 , 0 , 0
       0     .08       0   245.8    .045       0   260.8     .08       0
Bank Sta=245.8,260.8
XS Rating Curve= 0 ,0
Exp/Cntr=0.3,0.1

Type RM Length L Ch R = 1 ,13606.9 ,771.2,782.7,793.6
XS GIS Cut Line= 2
     1655750.578      320411.022     1656110.821      321031.682
#Sta/Elev= 30
       0  917.32    98.3  883.99   127.8  874.79   157.3  863.59     177  856.68
   186.8  852.78   196.6  847.72   226.1  831.07   235.9  826.78   245.8  824.36
   285.1  818.76   314.6  816.12   363.7   813.3     366  813.32   373.6  813.39
     381  814.48   383.4  814.84     403  822.26   412.9  824.37   422.7  825.58
   432.5   829.5   442.4  835.84   481.7  863.21   491.5   869.3   501.4  874.03
   540.7  890.55   570.2  903.43   658.6  943.97   688.1  956.78   717.6  968.75
#Mann= 3 , 0 , 0
       0     .06       0     366    .045       0     381      .1       0
Bank Sta=366,381
XS Rating Curve= 0 ,0
Exp/Cntr=0.3,0.1

Type RM Length L Ch R = 1 ,12824.2 ,469.2,469.2,469.1
XS GIS Cut Line= 2
     1655195.023      320402.342     1655221.089      321250.818
#Sta/Elev= 30
       0  926.63   107.3  892.33   156.1  874.39   165.9  870.08   185.4  859.47
   234.2  829.61   243.9  824.97   273.2  813.84   282.4  812.27     283  812.17
   297.4  812.51   331.7  815.08     361  816.52   419.6  818.36   468.4  818.72
   497.6  819.92   536.6  823.06     605  829.75   614.7  831.27   624.5  835.74
   673.2  869.99   692.8  881.29   702.5  888.04     722  905.28   731.8     913
   741.6  918.58   751.3  921.95   770.8   925.9   809.8  930.54   848.9  936.09
#Mann= 3 , 0 , 0
       0      .1       0   282.4    .045       0   297.4     .06       0
Bank Sta=282.4,297.4
XS Rating Curve= 0 ,0
Exp/Cntr=0.3,0.1

Type RM Length L Ch R = 1 ,12355   ,453.3,438.2,422.8
XS GIS Cut Line= 2
     1654736.844      320567.181     1654756.655       321161.89
#Sta/Elev= 30
       0  899.32    58.5  870.12    68.3  865.01    97.6   848.5   117.1  838.54
   126.8  834.02   146.3  825.65   175.6  814.14   185.3   811.3   195.1  810.47
   204.8  811.02   214.5  812.26   253.6  817.07   263.4  817.53   282.9  817.72
   302.4  818.92   312.2  818.81   321.9  820.07   341.4   828.4   360.9  832.39
   370.7  836.39   399.9  851.83   409.7  855.98   487.7   881.2   497.5  883.43
   507.2  884.23   546.3  883.65   575.5  883.61   585.3  882.62     595  880.83
#Mann= 3 , 0 , 0
       0      .1       0   175.6    .045       0   214.5     .06       0
Bank Sta=175.6,214.5
XS Rating Curve= 0 ,0
Exp/Cntr=0.3,0.1

Type RM Length L Ch R = 1 ,11916.8 ,480.1,463.1,445.8
XS GIS Cut Line= 4
     1654062.234      320515.141     1654220.654      320719.134
     1654511.453      321062.016     1654678.554      321183.544
#Sta/Elev= 30
       0  953.73    57.4  934.93      67  930.82    95.7  914.78   143.5   890.9
   200.9  868.65   258.3  841.83   287.6  832.68   297.4  831.38   316.9  829.99
     356     830   365.8  827.55   375.6  823.46   395.1  812.94   404.9  809.96
   424.4  811.05   473.3  815.45   580.8  814.67   619.9  816.76   639.5  820.12
   688.3  831.51   707.9  833.91   717.7  836.67   747.2  850.53   757.1  853.57
   796.4  861.41   816.1  864.84   845.6  867.92   875.1  874.84   914.5  871.98
#Mann= 3 , 0 , 0
       0      .1       0   395.1    .045       0   424.4     .06       0
Bank Sta=395.1,424.4
XS Rating Curve= 0 ,0
Exp/Cntr=0.3,0.1

Type RM Length L Ch R = 1 ,11453.7 ,233.1,232.9,232.4
XS GIS Cut Line= 3
     1653756.245      320992.571     1653993.787      321225.039
     1654576.557      321296.391
#Sta/Elev= 30
       0  914.86    39.1  910.19    97.8  904.96     176  899.91   205.3  900.11
   224.8  899.11   273.7   894.4   312.8  891.87   332.4  889.42   351.9  889.53
   361.7  888.35   371.5  883.23   381.3  874.14   420.4  831.14   430.2  822.35
     440  817.48   469.4  811.12   476.5  810.17   488.9  809.56   498.7  810.02
   547.6  813.74   606.4  817.22   694.4  820.99   704.2  821.96   733.6  827.73
   762.9  831.14   792.3  835.94   811.8  837.98     851  839.16   919.5  838.74
#Mann= 3 , 0 , 0
       0      .1       0   476.5    .045       0   498.7     .06       0
Bank Sta=476.5,498.7
XS Rating Curve= 0 ,0
Exp/Cntr=0.3,0.1

Type RM Length L Ch R = 1 ,11220.8 ,371.3,386.7,402.2
XS GIS Cut Line= 2
     1654029.377      321464.228     1654584.932      321522.822
#Sta/Elev= 30
       0   861.7     9.8  856.07    19.6  847.18    39.2  826.79      49  819.83
    58.8  816.94    78.4  814.46      98   811.2   107.8  809.89   117.6  809.95
   127.4  810.96   156.8  813.04     196  813.04   215.6  813.58   284.2  817.42
     294  818.73   303.8  821.54   323.4  828.81   333.2  831.11   352.8  833.82
   362.6  837.59   382.2   846.3   411.6  854.29   421.4   856.4   450.8  860.14
   480.2  861.14   509.6  863.74   529.2  864.76     539  865.93   558.6  869.76
#Mann= 3 , 0 , 0
       0      .1       0      98    .045       0   127.4     .06       0
Bank Sta=98,127.4
XS Rating Curve= 0 ,0
Exp/Cntr=0.3,0.1

Type RM Length L Ch R = 1 ,10834.1 ,68.3,68,67.6
XS GIS Cut Line= 3
     1653974.669       321339.36     1653981.614      321716.096
     1654325.967      322049.877
#Sta/Elev= 30
       0   872.7    19.3  869.99    77.3  867.19   125.6  864.09   164.2  864.98
   183.6  864.25   212.6  859.67   241.5  856.26   299.5   845.6   338.2  836.94
   386.6  824.51   406.2  820.27   425.7  818.67   464.9  817.64   484.5  816.52
     504  814.76     553  809.03   572.5  807.86   583.7  809.08   592.1  810.51
   611.7  815.38     641  826.38   650.8   828.7   660.6  834.42   680.2  851.93
     690  859.25   699.8   865.1   758.5  897.04   807.4  921.61   856.4  946.98
#Mann= 3 , 0 , 0
       0     .06       0     553    .045       0   583.7      .1       0
Bank Sta=553,583.7
XS Rating Curve= 0 ,0
Exp/Cntr=0.3,0.1

Type RM Length L Ch R = 1 ,10766.2 ,67,71.5,76
XS GIS Cut Line= 3
     1653750.711      321533.804     1653926.058      321756.026
     1654272.148      322086.335
#Sta/Elev= 30
       0  870.21    19.5  866.39    58.6  860.01   107.4  850.88   117.1  848.52
   156.2  840.85   195.2  831.32     205  829.31     244  826.85   273.3  823.69
   351.4  819.76   400.2  815.78   439.3   814.5   468.6   814.6   478.3     814
   488.1  812.07   497.9  809.52   507.6  807.99   517.4   808.6   527.2  810.78
   536.9  814.53   546.7   819.8   556.4  823.86   566.2  826.83     576  833.86
   595.5  854.32   605.3  862.21     615  867.89   673.6  899.69   761.5  943.67
#Mann= 3 , 0 , 0
       0     .06       0   497.9    .045       0   527.2      .1       0
Bank Sta=497.9,527.2
XS Rating Curve= 0 ,0
Exp/Cntr=0.3,0.1

Type RM Length L Ch R = 1 ,10694.7 ,67.3,72.8,78.1
XS GIS Cut Line= 3
     1653787.773      321610.641     1653917.378      321789.012
     1654195.155      322186.582
#Sta/Elev= 30
       0   859.9    28.8  856.08    47.9   852.5    95.9  841.16   105.4  838.48
     115  834.76   124.6  831.62   134.2  829.66   172.6  823.98   182.1  823.28
   220.5  822.36   249.6  821.05     269  819.44   298.1  815.84   317.5  813.85
   346.6  812.03   395.1  810.25   414.5  808.58   424.2  807.95   433.9  808.51
   443.6  810.69   453.3   814.9     463  819.98   482.4  826.07   492.1  831.49
   550.3  873.73   589.1  903.31   598.8  909.53   618.2  918.92   705.5  958.62
#Mann= 3 , 0 , 0
       0     .06       0   414.5    .045       0   443.6      .1       0
Bank Sta=414.5,443.6
XS Rating Curve= 0 ,0
Exp/Cntr=0.3,0.1

Type RM Length L Ch R = 1 ,10621.9 ,47.5,46.4,45.4
XS GIS Cut Line= 3
     1653537.169      321618.874     1653904.092      321818.974
     1654055.134      322207.863
#Sta/Elev= 30
       0  849.78    29.2  845.12    48.6  842.74   116.6  836.01   155.5  833.59
   233.3  825.91   281.9  823.68   320.7  824.42   359.6   821.5   417.9   821.2
     447  819.31   495.6  815.03   563.5  814.81   573.2  814.23   582.9  812.55
   592.6  809.97   602.3  808.13     612  808.38   621.7  810.17   641.1  817.83
   660.5  823.02   670.2  828.55   689.6  845.37     709   859.4   738.1  882.68
   786.6  916.51   796.3  921.34     806  924.45   825.4  929.03   835.1   930.5
#Mann= 3 , 0 , 0
       0     .06       0   592.6    .045       0   621.7      .1       0
Bank Sta=592.6,621.7
XS Rating Curve= 0 ,0
Exp/Cntr=0.3,0.1

Type RM Length L Ch R = 1 ,10575.4 ,98.1,96.7,95.4
XS GIS Cut Line= 3
     1653488.558       321683.11     1653863.558      321863.665
     1654028.489      322235.193
#Sta/Elev= 30
       0  881.85   154.9  843.94   183.9  838.79   222.6  833.96     271  825.81
   280.7  824.58     300   823.2   329.1  822.92   377.5  818.53   387.2  818.16
   416.2  818.63   435.6  817.51     484  813.59   551.7  810.34   571.1  808.13
   580.7  807.85   590.4  808.76   600.1  811.61   619.4   819.7   629.1  821.64
   638.8  825.36   648.5  831.95   658.2  839.64   696.9  872.74   706.6  880.64
   716.2  886.48   764.6  908.13     784  915.87   803.3   921.9   822.7  926.56
#Mann= 3 , 0 , 0
       0     .06       0   571.1    .045       0   590.4      .1       0
Bank Sta=571.1,590.4
XS Rating Curve= 0 ,0
Exp/Cntr=0.3,0.1

Type RM Length L Ch R = 1 ,10478.8 ,301.1,285.4,264.2
XS GIS Cut Line= 3
     1653471.197      321764.707       1653764.6      321903.596
      1653929.53       322223.04
#Sta/Elev= 30
       0  891.31    19.7  888.36    78.7  877.77   127.9  867.86   137.7  865.31
   157.4  858.96   177.1  851.49   216.4  839.52   245.9  828.89   255.8  826.46
   265.6  824.98   275.4  824.33   304.9  823.92   353.8   819.3   402.4  814.08
   460.6  810.88   480.1  808.94   489.8  808.04   499.5  808.11   505.7  809.09
   509.2  809.65   518.9   812.6   528.7  816.41   548.1  821.15   557.8  825.18
   616.1  862.75   645.3  880.24     655  884.93   664.7  888.32   684.1  893.34
#Mann= 3 , 0 , 0
       0     .06       0   480.1    .045       0   505.7      .1       0
Bank Sta=480.1,505.7
XS Rating Curve= 0 ,0
Exp/Cntr=0.3,0.1

Type RM Length L Ch R = 1 ,10193.3 ,258.5,261.2,269.3
XS GIS Cut Line= 3
     1653368.766      321950.471     1653740.748      322232.457
     1653940.401      322256.329
#Sta/Elev= 30
       0  924.15     9.7  921.45    19.4  916.89    29.2  910.78    58.4   891.2
     107  856.25   116.7  849.84   126.4  845.04     175  823.48   204.2  812.46
   213.9  809.58   223.7  807.67   245.6  805.95   262.6   805.8   272.3   805.8
   311.2  807.67   320.9   806.6   330.6  806.46   369.5  815.28   379.3  816.85
     389  817.66   408.4  818.17   447.3  818.18   457.1  819.22   466.8  821.03
   485.9  827.15   514.7   838.1     620  882.66   639.1  889.66   667.9  898.81
#Mann= 3 , 0 , 0
       0      .1       0   245.6    .045       0   272.3     .06       0
Bank Sta=245.6,272.3
XS Rating Curve= 0 ,0
Exp/Cntr=0.3,0.1

Type RM Length L Ch R = 1 ,9932.1  ,258.2,255.8,253.4
XS GIS Cut Line= 2
      1653170.85      322141.443     1653754.183      322479.985
#Sta/Elev= 30
       0  919.67    48.9  919.01    58.6  918.51    68.4  916.63    78.2  912.06
      88  905.76   117.3   884.3   156.4  854.67   166.2  847.99   175.9  842.62
   234.6   811.9   244.4  807.36   250.2  806.55   254.1  806.01   263.9   805.8
   273.7  805.94   283.5  806.64   322.6  810.86   381.2  815.55   439.9  818.92
   498.5  823.51   508.3  823.94   527.8  823.68   547.4  822.36   566.9  820.47
   576.7  820.51   596.3   822.6   615.8  823.85   645.1  826.41   674.4   828.2
#Mann= 3 , 0 , 0
       0      .1       0   250.2    .045       0   273.7     .06       0
Bank Sta=250.2,273.7
XS Rating Curve= 0 ,0
Exp/Cntr=0.3,0.1

Type RM Length L Ch R = 1 ,9676.3  ,347.5,347.4,347.3
XS GIS Cut Line= 2
     1652957.362      322355.063     1653580.337       322632.61
#Sta/Elev= 30
       0  861.62    19.5  859.88    29.2  860.19    68.2  864.53   116.9  871.34
   126.7  871.59   175.4  870.39   204.6  867.95   214.3  866.25   224.1  863.49
   253.3     851   263.1  846.13     302  824.74   321.5  812.72   332.1  807.57
     341  805.89   360.5  806.41   409.2  810.01   526.1   814.7   535.9  815.35
   545.6  816.89   555.4  819.57   584.6  829.31   594.3  831.47   604.1  832.63
   613.8  835.12     643   848.4   652.8  852.18   672.3   858.5     682   860.7
#Mann= 3 , 0 , 0
       0      .1       0   332.1    .045       0   360.5     .06       0
Bank Sta=332.1,360.5
XS Rating Curve= 0 ,0
Exp/Cntr=0.3,0.1

Type RM Length L Ch R = 1 ,9328.9  ,237.4,250.8,264.1
XS GIS Cut Line= 2
     1653049.569      322776.036     1653440.194      322937.494
#Sta/Elev= 30
       0  849.16     9.8  845.91    19.7  841.38    39.3  831.36    68.8  815.83
    78.6  810.94    88.5  807.44    98.3  805.99   116.7   805.8     118   805.8
   127.8  805.85   137.6  806.24   167.1  808.49   176.9     809   186.8  809.32
   226.1  810.07   245.7   810.8   265.4  811.93   275.2  812.85   285.1  815.47
   294.9  819.98   304.7   824.7   314.6  827.93   324.4  829.68   334.2  832.01
     344  835.62   363.7  843.46   383.4  851.53   412.8  864.29   422.7  868.46
#Mann= 3 , 0 , 0
       0      .1       0    98.3    .045       0     118     .06       0
Bank Sta=98.3,118
XS Rating Curve= 0 ,0
Exp/Cntr=0.3,0.1

Type RM Length L Ch R = 1 ,9078.1  ,49.2,48.8,48.5
XS GIS Cut Line= 3
     1652973.537      322867.585     1653158.697      323146.651
     1653456.176      323273.835
#Sta/Elev= 30
       0  840.32     9.6  838.67    19.1  836.48    47.8  829.11   114.8  809.43
   124.4  807.85     134   807.7   172.2  809.76   181.8  808.98   191.4  807.24
   200.9  806.01   210.5  805.82   220.1  806.38   229.6  808.36   239.2  809.48
   258.4  811.24   277.5  813.71   306.2  815.98   344.7  822.54   364.3  823.92
   374.1  825.54   393.7  830.68   413.3  835.22   432.9  841.58   452.6  849.21
     482  861.53   540.8  887.16   560.4  895.02   609.4  912.35   658.4   930.5
#Mann= 3 , 0 , 0
       0     .06       0   191.4    .045       0   220.1     .06       0
Bank Sta=191.4,220.1
XS Rating Curve= 0 ,0
Exp/Cntr=0.3,0.1

Type RM Length L Ch R = 1 ,9029.2  ,133.5,136.7,139.7
XS GIS Cut Line= 3
     1652911.037      322867.585     1653115.898      323166.196
      1653119.37      323419.668
#Sta/Elev= 30
       0  840.51    29.4  836.08    58.7   832.2    68.5  830.43   127.2  814.46
   146.8  810.36   156.6  808.77   166.4  807.85   176.2  807.93   205.5  809.52
   215.3   809.1   225.1   807.1   234.9  805.94   244.7  806.68   254.5  809.28
   264.3  810.67   283.8  809.64   293.6  810.18   303.4  811.39   332.8  815.95
   362.1  819.74   391.4  821.08   401.1  823.03   410.9  827.37   440.1  846.13
   479.1  870.56   547.4  911.33   566.9  921.77   596.1  935.81   615.6  946.22
#Mann= 3 , 0 , 0
       0     .06       0   225.1    .045       0   244.7     .06       0
Bank Sta=225.1,244.7
XS Rating Curve= 0 ,0
Exp/Cntr=0.3,0.1

Type RM Length L Ch R = 1 ,8892.6  ,254.3,267.9,281.6
XS GIS Cut Line= 2
     1652848.769      322975.161     1653044.082      323354.935
#Sta/Elev= 30
       0  830.16     9.7  828.54    19.4  826.07    38.8  819.94    48.5  817.17
    58.2  814.81    67.9  813.01    77.6  811.57    87.4  810.41    97.1  809.45
   106.8  808.56   126.2  807.06   145.6  806.03   155.3  805.82     165   805.8
   194.1  805.81   203.8  806.23   213.5  807.15   242.6  810.48   281.5  815.24
   300.9  817.42   310.6   818.2   320.3  818.69     330  820.78   339.7  826.42
   349.4   833.1   378.5   854.1   407.6  875.43   417.4  882.49     427   889.6
#Mann= 3 , 0 , 0
       0     .06       0     165    .045       0   194.1     .06       0
Bank Sta=165,194.1
XS Rating Curve= 0 ,0
Exp/Cntr=0.3,0.1

Type RM Length L Ch R = 1 ,8624.6  ,370.2,401.3,432.3
XS GIS Cut Line= 3
     1652977.141      322695.744     1652742.766      323082.029
     1652703.703      323537.758
#Sta/Elev= 30
       0  861.13    88.4  850.96   127.7  849.17     167  843.28   196.4  839.71
   294.7  833.89     334  830.45   353.6  827.81   422.4  816.53   461.6   808.5
   471.3  807.45   549.2   805.8   597.8  805.81   617.3  806.16     627  808.03
   646.5   814.4   665.9  817.94   675.7  822.42   685.4   829.3   704.9   844.7
   743.8  876.55   763.2   891.8   782.7  905.43   792.4  911.52   811.9  922.14
   821.6  925.91   831.4  928.44   860.6  931.74   899.5  943.11   909.2  947.64
#Mann= 3 , 0 , 0
       0     .06       0   597.8    .045       0   617.3      .1       0
Bank Sta=597.8,617.3
XS Rating Curve= 0 ,0
Exp/Cntr=0.3,0.1

Type RM Length L Ch R = 1 ,8223.3  ,906.2,882.7,858.8
XS GIS Cut Line= 3
     1652856.378      322138.165       1652705.5      322981.577
     1652330.337      323025.318
#Sta/Elev= 30
       0     908      39  887.96    77.9  865.79    97.4  859.23   116.8  855.43
     146  851.48   204.5  845.75   262.9  838.36   282.4  834.65   311.6  826.48
   340.8  822.15     370   820.5   399.2  821.56   447.9  818.75   632.9  822.34
   808.1   822.1   856.8   820.1   876.2  817.17   914.9  809.11   934.3  806.74
   992.4  805.36  1031.1     807  1069.9  804.62  1098.9  804.08  1118.3  804.25
  1137.1     806    1157   813.3  1176.4  817.13  1186.1  822.46  1234.5   858.3
#Mann= 3 , 0 , 0
       0     .06       0  1118.3    .045       0  1137.1      .1       0
Bank Sta=1118.3,1137.1
XS Rating Curve= 0 ,0
Exp/Cntr=0.3,0.1

Type RM Length L Ch R = 1 ,7340.7  ,616.1,583.6,551.1
XS GIS Cut Line= 4
     1652794.982      321891.009     1652554.096      322338.058
     1652406.527      322546.391     1652308.738      323016.925
#Sta/Elev= 30
       0  983.44    29.3  980.72    48.8  976.29    68.4  969.15    87.9  958.82
   117.2  941.56   146.5  922.51   224.6  867.47   263.7  841.11   322.3   805.2
     332   800.6   341.8  799.39   361.3  801.47   380.9  804.44   400.4  806.16
   429.7  807.37   576.6  817.37   694.4  818.45   900.4   818.5   939.7  819.06
   978.9  822.12  1008.3  821.85  1018.1  822.82  1027.9  825.02  1057.4  835.86
  1096.6  845.43  1165.2  855.98  1184.9  860.25  1214.3  864.59  1243.7  870.32
#Mann= 3 , 0 , 0
       0      .1       0     332    .045       0   361.3     .06       0
Bank Sta=332,361.3
XS Rating Curve= 0 ,0
Exp/Cntr=0.3,0.1

Type RM Length L Ch R = 1 ,6757.1  ,488.6,485.9,483.2
XS GIS Cut Line= 3
     1651792.378      322186.148     1652371.805      322609.325
     1652289.339       323004.29
#Sta/Elev= 30
       0   984.3    68.8  955.24   108.1  935.55     118  929.97   127.8  923.24
   147.4  908.37   167.1  894.86   176.9  890.25   196.6  885.86   265.4  873.62
   304.7  862.43   324.4  854.32     403  807.76   412.8  802.27   422.6  799.24
   432.5  798.81   450.7  799.37   520.9  801.54   589.7  804.75   678.2  811.28
   717.5  815.29   806.1  817.58   855.3  821.44   894.6  821.99   914.3   825.3
   943.8  834.57   953.7  836.66  1002.9  843.64  1052.1  852.97    1121  862.52
#Mann= 3 , 0 , 0
       0      .1       0   422.6    .045       0   450.7     .06       0
Bank Sta=422.6,450.7
XS Rating Curve= 0 ,0
Exp/Cntr=0.3,0.1

Type RM Length L Ch R = 1 ,6271.2  ,203.6,203.6,203.7
XS GIS Cut Line= 2
     1651787.037      322797.654     1652262.731      323065.015
#Sta/Elev= 30
       0  889.66    19.5  876.54    68.2  843.18    87.7  830.33   107.2  818.02
   116.9  811.54   126.7  804.25   130.6  801.99   136.4  798.63   146.2  797.67
   155.9  797.92   165.6  798.62   194.9  800.81   214.4  801.82   253.4  803.06
   321.6  803.73   360.5  804.74     380   805.4   389.8  806.04   399.5  807.46
   409.3  810.17     419  813.49   428.8  816.48   438.5  818.29   448.2  819.78
     458  822.63   467.7  827.04   477.5  831.94   506.7  846.78   545.7  866.98
#Mann= 3 , 0 , 0
       0      .1       0   130.6    .045       0   165.6     .06       0
Bank Sta=130.6,165.6
XS Rating Curve= 0 ,0
Exp/Cntr=0.3,0.1

Type RM Length L Ch R = 1 ,6067.5  ,512.2,520.4,528.5
XS GIS Cut Line= 3
     1651716.878      322936.972     1651798.476      323032.459
     1652178.684         323246.
#Sta/Elev= 30
       0  864.72    38.6  845.38      58  836.19    77.3  827.56    96.6  819.73
   115.9  812.65   125.6  809.41   164.4  798.15   173.3  796.44   183.7  795.58
   193.4  795.76   203.1  796.33     271  800.58     300  803.14   319.4  805.57
   348.5  810.91   358.2  812.24   367.9  813.18   377.6  813.52   387.2  813.32
   396.9  812.32   406.6  812.69   416.3  815.33     426  817.42   435.7  818.63
   445.4  820.45   455.1  823.54   503.5  840.61   532.6  851.13   561.7  861.07
#Mann= 3 , 0 , 0
       0      .1       0   173.3    .045       0   203.1     .06       0
Bank Sta=173.3,203.1
XS Rating Curve= 0 ,0
Exp/Cntr=0.3,0.1

Type RM Length L Ch R = 1 ,5547.2  ,504.8,496.1,486.1
XS GIS Cut Line= 2
     1651373.739      323157.262     1651859.953       323734.46
#Sta/Elev= 30
       0  847.81    39.2  837.09   117.6  818.46   156.8  807.92   166.6  805.88
   176.4  804.59   235.2  799.83   274.4  797.73   303.8  797.43   352.8  797.44
   431.2  798.21   450.9  797.65   470.5   796.7   499.9  794.33   509.7   793.5
   519.5  793.27   529.3  794.39   548.9  798.56   558.7   800.9   568.5  804.03
   588.1  808.37   597.9  812.47   607.7  818.71   617.5  825.54   646.9  847.02
   666.5  860.68   686.1  873.72   725.3  899.12   744.9  912.96   754.7  919.49
#Mann= 3 , 0 , 0
       0     .06       0   499.9    .045       0   529.3      .1       0
Bank Sta=499.9,529.3
XS Rating Curve= 0 ,0
Exp/Cntr=0.3,0.1

Type RM Length L Ch R = 1 ,5051.1  ,573.4,553.8,535.4
XS GIS Cut Line= 4
     1650674.756      323590.228     1651117.464       323618.44
      1651462.57      323813.397     1651819.341      323857.667
#Sta/Elev= 30
       0 1039.09    67.5 1001.67   125.4  970.86   154.3  954.81   192.9  932.68
   241.1  904.12   260.4  895.02   318.2  871.85   424.3  831.02   501.6  809.83
   569.3  794.42     579  792.75   598.3  792.21     608  792.39   675.6   795.9
   733.6  801.51   743.3  802.74   762.6   807.6   772.3  808.93     782   811.4
   791.6  816.35     811  828.97   820.6  834.01   830.3  838.02   937.1  866.24
   966.3  876.08  1005.2  891.73    1044   906.2  1092.6     919  1199.5  950.77
#Mann= 3 , 0 , 0
       0      .1       0   569.3    .045       0     608     .06       0
Bank Sta=569.3,608
XS Rating Curve= 0 ,0
Exp/Cntr=0.3,0.1
